HEC-RAS study A119-00-00.prj: A119-00-00

--- A119-00-00.g01 (geometry) --- (continued)

Type RM Length L Ch R = 1 ,16142.95,118.54,121.38,120.01
BEGIN DESCRIPTION:
Astoria Blvd
END DESCRIPTION:
XS GIS Cut Line= 6
      3178878.23    13782813.437     3178463.977    13782399.098
      3178360.45     13782303.83     3177011.415    13780928.958
     3175667.033     13779599.73     3175090.285    13778978.609
#Sta/Elev= 30
  4223.7   27.73  4346.7    32.1 4455.72    32.7 4498.14   28.55 4540.56   27.74
  4942.4   27.73 4964.96   22.75    4977   12.85    5045   12.85 5049.56   20.43
  5065.8   26.14 5089.86   28.34 5475.74   27.02 5949.68   29.36 6322.72    27.4
 6491.48   29.23 6584.22   27.68 6704.74   29.97 6909.24   28.55 6959.02   31.03
 7164.81   28.62 7210.78   30.53 7454.76   30.72 7867.36   28.31 8125.19   30.77
 8199.43   28.68 8289.19   31.15 8522.13   29.58  8698.2   31.06 9614.67   30.47
#Mann= 4 ,-1 , 0
  4223.7     .07       0  4942.4    .015       0 5089.86     .15       0
  8698.2     .07       0
#XS Ineff= 3 ,-1
    7000    8700      30    4300    4977   28.75    5043    6999      28
Permanent Ineff=
       F       F       F
#Block Obstruct= 1 ,-1
 4175.82 4455.11    32.7
Bank Sta=4942.4,5089.86
XS Rating Curve= 0 ,0
Exp/Cntr=0.5,0.3

Type RM Length L Ch R = 2 ,16081   ,,,
BEGIN DESCRIPTION:
Culverts at Astoria Blvd
END DESCRIPTION:
Bridge Culvert--1,0,-1,-1, 0
Deck Dist Width WeirC Skew NumUp NumDn MinLoCord MaxHiCord MaxSubmerge Is_Ogee
4,101,2.6,0, 15, 15, , , 0.95, 0, 0,0,,
    4225    4325    4483    4570    4820    4870    4920    4955    4955    5065
    5065    5113    5175    5304    6872
   27.81   30.87   30.55    27.9   28.35   28.69   28.99   28.99   29.43   29.43
   29.31   29.12   28.65   27.41   28.98
       0       0       0       0       0       0       0       0       0       0
       0       0       0       0       0
    4225    4325    4483    4570    4820    4870    4920    4955    4955    5065
    5065    5113    5175    5304    6872
   27.81   30.87   30.55    27.9   28.35   28.69   28.99   28.99   29.43   29.43
   29.31   29.12   28.65   27.41   28.98
       0       0       0       0       0       0       0       0       0       0
       0       0       0       0       0
Culvert=2,12,10,101,0.012,0.5,1,10,1,13.06,4988.5,12.99,4988.5,Culvert #1  , 0 ,4
Culvert Bottom n=0.012
Culvert=2,12,10,101,0.012,0.5,1,10,1,13.01,4999.5,13.01,4999.5,Culvert #2  , 0 ,4
Culvert Bottom n=0.012
Culvert=2,12,10,101,0.012,0.5,1,10,1,13.09,5010,12.99,5010,Culvert #3  , 0 ,4
Culvert Bottom n=0.012
Culvert=2,12,10,101,0.012,0.5,1,10,1,13.07,5020.5,12.88,5020.5,Culvert #4  , 0 ,4
Culvert Bottom n=0.012
Culvert=2,12,10,101,0.012,0.5,1,10,1,13.03,5031.5,12.94,5031.5,Culvert #5  , 0 ,4
Culvert Bottom n=0.012
BC Design=,, 0 ,, 0 ,,,,,,
BC HTab HWMax=32.7
BC Use User HTab Curves=0
BC User HTab FreeFlow(D)= 0

Type RM Length L Ch R = 1 ,16021.58,81.59,80.04,80.03
BEGIN DESCRIPTION:
Astoria Blvd
END DESCRIPTION:
XS GIS Cut Line= 6
      3178972.18     13782742.97     3178548.244    13782313.647
     3178352.605    13782124.791     3177451.725    13781200.302
     3175842.345    13779615.674     3175180.877    13778911.504
#Sta/Elev= 30
 4212.94   27.93 4364.32   32.24 4459.93   31.95 4491.19   29.09 4934.41   28.85
  4965.7   24.12    4977   12.85    5045   12.85 5048.43   17.83 5058.45   22.26
 5097.25   28.53 5226.46   26.85 5378.53   28.72 5486.81   26.72 5721.57   29.08
 6056.72   27.66 6249.31    29.7  6338.4   27.66 6406.82   29.85 6545.47   29.73
 6604.98   27.72 7103.51   29.99 7418.39   28.45 7683.94   30.66 7822.62   30.61
 7902.42   28.14 8023.18   31.07 8218.36   28.96 8579.51   31.19 9603.76   30.66
#Mann= 4 ,-1 , 0
 4212.94     .07       0 4934.41    .015       0 5097.25     .15       0
 8579.51     .07       0
#XS Ineff= 3 ,-1
    7700    8600      30    4350    4977   28.75    5043    7575      28
Permanent Ineff=
       F       F       F
#Block Obstruct= 1 ,-1
 4174.31 4363.84   32.23
Bank Sta=4934.41,5097.25
XS Rating Curve= 0 ,0
Exp/Cntr=0.5,0.3

Type RM Length L Ch R = 1 ,15941.54,334.52,332.61,344.22
BEGIN DESCRIPTION:
Astoria Blvd
END DESCRIPTION:
XS GIS Cut Line= 6
      3179034.82    13782688.162     3178604.422     13782256.68
     3178409.167    13782068.206     3177508.568    13781144.006
     3175963.015    13779609.032     3175241.272     13778857.82
#Sta/Elev= 30
 4210.18   27.83 4344.65   31.85 4612.39    28.1 4925.74   30.32  4954.5   26.83
 4977.77   19.48    4982   12.85    5037   12.85 5041.48   17.32 5058.16   23.26
 5088.59   28.19 5769.98   27.35 5990.22   29.49 6062.66   26.98 6128.12    29.5
 6331.46   27.45  6498.6   30.14  6615.6   27.83  6757.5   30.62 6903.34   27.99
 6955.04   30.47 7193.36   30.94 7418.05    28.1 7463.77   30.32 7856.56   30.74
 7923.25   28.01 8024.76   31.15 8236.54   29.09 8469.29   31.21 9601.46   30.82
#Mann= 4 ,-1 , 0
 4210.18     .07       0 4925.74    .015       0 5088.59     .15       0
 8469.29     .07       0
#XS Ineff= 1 ,-1
    7200    8500      30
Permanent Ineff=
       F
#Block Obstruct= 1 ,-1
 4185.99 4343.87   31.83
Bank Sta=4925.74,5088.59
XS Rating Curve= 0 ,0
Exp/Cntr=0.3,0.1

Type RM Length L Ch R = 1 ,15608.93,606.91,597.34,549.72
XS GIS Cut Line= 6
      3179261.88    13782445.441     3178778.484     13781955.37
     3178658.669    13781849.224     3177418.246    13780541.248
     3176594.899    13779649.447       3175572.6    13778591.813
#Sta/Elev= 30
 4223.63   27.69 4263.52   26.03  4296.5   31.22 4334.52   32.44 4428.26   32.12
 4482.08      28  4535.9   27.51 4709.83   30.69 4905.14   31.32 4929.52    29.3
 4949.36   28.13  4995.6   13.62 5020.07   13.82 5050.64   29.53 5055.45   29.72
 5780.99    27.7 5959.53   29.99 6343.39      28 6444.67    30.1 6802.82   30.63
 6892.59   28.43 6949.07   30.52  7346.7   30.67 7474.83   27.85 7633.99   30.63
 8012.09   30.55 9112.12   30.97 9156.31   28.66 9206.67   30.94 9559.48   30.76
#Mann= 4 ,-1 , 0
 4223.63     .07       0 4929.52    .015       0 5055.45     .15       0
 8012.09     .07       0
#XS Ineff= 2 ,-1
    4400    4800      30    5150    7700      30
Permanent Ineff=
       F       F
#Block Obstruct= 2 ,-1
  4161.4 4333.83   32.41 9056.93 9621.64      30
Bank Sta=4929.52,5055.45
XS Rating Curve= 0 ,0
Exp/Cntr=0.3,0.1

Type RM Length L Ch R = 1 ,15011.6 ,100.37,96.59,111.89
XS GIS Cut Line= 6
      3179725.32    13782035.953     3179174.266    13781513.937
      3179088.71    13781434.085     3178032.325    13780506.363
     3177575.796    13780360.803      3175722.11    13778469.482
#Sta/Elev= 30
 4191.29   20.32 4211.04   28.74 4301.56   32.76 4431.19   32.02 4499.41   28.11
 4639.53   31.05 4887.45    31.6  4942.6   29.75 4964.36   28.13 5004.22   13.86
  5010.6   13.62 5035.07   13.82 5065.64   29.53 5070.45   29.72 5204.48    30.1
 5273.39   27.67 5418.14   29.72 5468.29   27.34 5581.34   29.47 5780.01   27.53
 6020.53   29.63 6156.96   27.26 6559.35   29.96 6946.26   27.78  7869.7   31.01
 8671.12   30.48 9118.75   26.52  9495.3   32.46 9545.63   29.13 9600.72   29.85
#Mann= 4 ,-1 , 0
 4191.29     .07       0  4942.6    .015       0 5070.45     .15       0
  7869.7     .07       0
#XS Ineff= 2 ,-1
    4390    4875      31    5160    7300      30
Permanent Ineff=
       F       F
#Block Obstruct= 2 ,-1
 4140.74 4360.72   33.17  7912.7 9699.15      30
Bank Sta=4942.6,5070.45
XS Rating Curve= 0 ,0
Exp/Cntr=0.3,0.1

Type RM Length L Ch R = 1 ,14915.01,1501.32,1223.07,424.92
XS GIS Cut Line= 6
      3179790.47    13781957.088     3179239.584    13781443.626
     3178989.211     13781205.44     3178093.633    13780420.419
     3177629.584     13780296.12     3175798.236    13778408.581
#Sta/Elev= 30
 4200.81   28.96 4328.81   33.12 4516.75   28.44 4649.04   30.65 4906.77   31.47
  4927.6   29.75 4964.36   28.13 5004.22   13.86  5010.6   13.62 5035.07   13.82
 5065.64   29.53 5070.45   29.72 5201.59    29.8 5450.88   27.18 5672.33   29.68
 5763.27   27.42 5977.15   29.64 6162.61   27.44 6240.33   29.65 6490.18    30.1
 6641.15    27.5  6805.7   29.69 6963.76   27.67 7028.44   30.23 7764.77   30.19
 8761.01   30.83 8976.53   27.69 9050.74   30.97  9428.1   28.92 9600.75   30.24
#Mann= 5 ,-1 , 0
 4200.81     .07       0  4927.6    .015       0 5070.45     .07       0
 5201.59     .15       0 7764.77     .07       0
#XS Ineff= 2 ,-1
    4390    4800      31    5150    7700   29.75
Permanent Ineff=
       F       F
#Block Obstruct= 2 ,-1
 4167.79 4328.62   33.12 8850.49 9633.82   29.74
Bank Sta=4927.6,5070.45
XS Rating Curve= 0 ,0
Exp/Cntr=0.3,0.1

Type RM Length L Ch R = 1 ,13691.93,22.52,20.62,21.09
BEGIN DESCRIPTION:
Ryewater Drive
END DESCRIPTION:
XS GIS Cut Line= 6
      3180829.49    13780909.709     3180320.298    13780446.538
     3179598.554     13780417.75     3179443.735    13780414.773
      3177660.95    13780261.552     3175843.912    13778367.981
#Sta/Elev= 30
 3645.71   30.44 3742.88   33.04 3848.56   30.11 4193.66   28.54 4252.46    30.5
  4339.6    27.5 4458.92   32.16 4598.88   30.08 4733.76   33.11 4952.11   27.62
 4976.02    14.8  4996.8   12.78 5024.52   16.55 5047.89   27.62 5803.48   29.49
 5966.82   27.86 6129.52   29.73 6240.64   27.64 6330.12   29.66  6709.1      30
 6801.38   27.37 6951.82   27.36 7053.73   30.31 7711.58   30.02 8846.36   31.08
 9008.69   27.72 9091.92   30.77 9531.14   32.25 9556.48   30.02 9624.93   29.59
#Mann= 5 ,-1 , 0
 3645.71     .07       0 4952.11    .015       0 5047.89     .07       0
 5803.48     .15       0 7711.58     .07       0
#XS Ineff= 2 ,-1
 3780.43 4736.06      31    5850    8000   29.65
Permanent Ineff=
       F       F
#Block Obstruct= 2 ,-1
 3597.07 3743.05   33.05 8867.62 9709.67    29.6
Bank Sta=4952.11,5047.89
XS Rating Curve= 0 ,0
Exp/Cntr=0.5,0.3

Type RM Length L Ch R = 1 ,13671.31,78.82,71.69,73.82
BEGIN DESCRIPTION:
Ryewater Drive
END DESCRIPTION:
XS GIS Cut Line= 6
      3180842.95    13780894.914     3180328.367    13780426.841
     3179694.865    13780401.794     3179444.785    13780394.789
     3177698.391    13780244.696     3175875.939    13778350.623
#Sta/Elev= 30
 3622.98   30.43 3721.64   33.07 3822.66   30.15 4182.96   28.22 4246.64   30.64
 4391.18   30.72 4499.14   28.24 4900.96   29.66 4952.11   27.62 4976.02    14.8
  4996.8   12.78 5024.52   16.55 5047.89   27.62 5092.88   29.22 5387.42   27.22
    5512   29.58  5789.3   29.49 5963.72    27.8 6121.28   29.72  6238.3   27.67
 6326.28   29.66  6691.2      30  6905.6   27.19  7021.5   30.38 7676.54   29.53
 8844.52   31.15 8996.35   27.75 9069.78   30.66 9498.65   32.03 9584.09   28.87
#Mann= 5 ,-1 , 0
 3622.98     .07       0 4952.11    .015       0 5047.89     .07       0
  5789.3     .15       0 7676.54     .07       0
#XS Ineff= 4 ,-1
    3771 4390.86   30.64    4392    4950    28.5    5050    5780    28.5
    5781    7900   29.65
Permanent Ineff=
       F       F       F       F
#Block Obstruct= 2 ,-1
 3594.27  3721.2   33.06 8868.11 9693.52    29.6
Bank Sta=4952.11,5047.89
XS Rating Curve= 0 ,0
Exp/Cntr=0.5,0.3

Type RM Length L Ch R = 3 ,13635   ,,,
BEGIN DESCRIPTION:
Bridge at Ryewater Drive
END DESCRIPTION:
Bridge Culvert--1,0,-1,-1, 0
Deck Dist Width WeirC Skew NumUp NumDn MinLoCord MaxHiCord MaxSubmerge Is_Ogee
3,52,2.6,0, 14, 14, , , 0.95, 0, 0,0,,
    4424    4798    4848    4904    4950    4950    4956    5000    5050    5050
    5052    5097    5150    5307
   29.57   28.97    29.3   29.54   29.52   29.83   29.83   29.83   29.83   29.68
   29.53   29.45   29.11   27.68
       0       0       0       0       0   27.77   27.77   27.77   27.77       0
       0       0       0       0
    4424    4798    4848    4904    4950    4950    4956    5000    5050    5050
    5052    5097    5150    5307
   29.57   28.97    29.3   29.54   29.52   29.83   29.83   29.83   29.83   29.68
   29.53   29.45   29.11   27.68
       0       0       0       0       0   27.77   27.77   27.77   27.77       0
       0       0       0       0
Pier Skew, UpSta & Num, DnSta & Num=  ,4985, 4 ,4985, 4 , 3 , 3 , 0 ,,
    1.15    1.15       2       2
       0   25.77   25.77      28
    1.15    1.15       2       2
       0   25.77   25.77      28
Pier Skew, UpSta & Num, DnSta & Num=  ,5015, 4 ,5015, 4 , 3 , 3 , 0 ,,
    1.15    1.15       2       2
       0   25.77   25.77      28
    1.15    1.15       2       2
       0   25.77   25.77      28
BR Coef=-1 , 1 , 0 ,, 0 ,,,0.8,-1,2,0,
WSPro=,,,, 1 ,,,, 0 ,,,, 0 ,,,,-1 ,-1 ,-1 , 0 , 0 , 0 , 0 , 0
BC Design=,, 0 ,, 0 ,,,,,,
BC HTab HWMax=33.07
BC Use User HTab Curves=0
BC User HTab FreeFlow(D)= 0

Type RM Length L Ch R = 1 ,13599.62,90.07,80.68,84.37
BEGIN DESCRIPTION:
Ryewater Drive
END DESCRIPTION:
XS GIS Cut Line= 6
      3180890.05    13780843.131     3180356.608    13780357.903
     3179601.316    13780327.786     3179448.459    13780324.847
     3177814.727    13780184.437     3175957.242     13778269.32
#Sta/Elev= 30
 3566.07   30.38 3668.04   33.15 3757.16   30.29 4135.92   29.64 4171.82   27.85
 4261.18   30.59  4342.4   27.96 4384.64   30.43 4507.52   28.89 4836.86   30.11
 4952.11   27.62 4976.02    14.8  4996.8   12.78 5009.08    13.1 5024.52   16.55
 5047.89   27.62 5393.98   30.14 5890.26   29.53 5971.44   27.57 6117.56   29.69
 6251.44   27.85 6440.32   29.39 6746.32   27.05 6900.19   29.83 7425.51   29.75
 7959.89   30.41 8835.57   31.11 8949.12   29.12 9389.14   30.81 9503.67   28.48
#Mann= 6 ,-1 , 0
 3566.07     .07       0 4952.11    .015       0 5047.89     .07       0
 5890.26     .15       0 7425.51     .12       0 7959.89     .07       0
#XS Ineff= 5 ,-1
 3714.79 4384.04    30.5    4600    4950    28.5    5050    5450    28.5
    4400    4550    29.5    5451    7850    29.5
Permanent Ineff=
       F       F       F       F       F
#Block Obstruct= 2 ,-1
 3533.27 3667.27   33.15 8893.09 9584.35    29.6
Bank Sta=4952.11,5047.89
XS Rating Curve= 0 ,0
Exp/Cntr=0.5,0.3

Type RM Length L Ch R = 1 ,13518.95,89.41,500.05,1112.06
BEGIN DESCRIPTION:
Ryewater Drive
END DESCRIPTION:
XS GIS Cut Line= 6
      3180943.88    13780783.951     3180388.884    13780279.117
     3179603.771    13780247.819     3179452.658    13780244.913
     3177870.746    13780108.956     3175841.094    13777967.335
#Sta/Elev= 30
 3518.34   31.16  3617.4   33.15 3704.03   30.55 4039.12   30.16 4169.83   28.23
 4237.71   30.85 4283.61   30.44 4351.69   26.69 4388.69   30.31 4433.73   29.17
 4529.94   31.57 4765.03   31.84 4952.11   27.62 4976.02    14.8  4996.8   12.78
 5009.08    13.1 5024.52   16.55 5047.89   27.62 5314.32   30.17 5835.86   28.97
 5945.65    29.4 6015.39   27.16 6130.02   29.43 6591.48   28.19 6767.77   29.65
 6862.66   27.58 6983.72   29.95 7253.63   29.91 7315.88   29.31 9743.82   29.05
#Mann= 6 ,-1 , 0
 3518.34     .07       0 4952.11    .015       0 5047.89     .07       0
 5835.86     .15       0 7253.63     .07       0 7315.88     .12       0
#XS Ineff= 2 ,-1
 3621.16 4544.94    30.5    5400    7800    29.6
Permanent Ineff=
       F       F
#Block Obstruct= 2 ,-1
 3487.74    3617   33.15  9487.5 9822.95    29.6
Bank Sta=4952.11,5047.89
XS Rating Curve= 0 ,0
Exp/Cntr=0.3,0.1

Type RM Length L Ch R = 1 ,13018.9 ,25.52,50,317.37
BEGIN DESCRIPTION:
Added cross-section is interpolated in channel banks and uses 2001 LiDAR in the overbanks and survey in the project boundary
Watearth, 2018
END DESCRIPTION:
XS GIS Cut Line= 6
 3180975.959577613780763.0775837 3180437.875451113780215.7620929
 3180173.599818313780019.6633645 3179719.187528813779664.5657316
 3178511.116944913778703.2600368 3176125.7665147 13776070.652071
#Sta/Elev= 30
 3552.38   30.02 3736.78   30.05 3781.64   38.22 4000.93   30.05 4294.98   31.09
 4454.53   26.04 4777.35      31  4912.3   26.34 4933.46   12.31  4993.4   11.88
 5033.94   13.12 5074.92   26.39 5235.84   30.29 5280.81   25.15 5405.72   29.53
 6105.21    25.7 6689.78   31.36  7224.7   31.83  7319.7   27.87 7444.69   31.84
    7555   28.59 7590.81    17.5 7764.75    17.5    7800   29.25    8785    28.5
    8812    19.5    9123    19.5    9150    28.510270.75   30.8510322.26   28.59
#Mann= 9 ,-1 , 0
 3552.38     .07       0  4912.3    .015       0 5074.92     .07       0
 6689.78     .12       0    7555    .012       0    7800     .12       0
    8785    .012       0    9150     .12       010270.75     .07       0
#XS Ineff= 2 , 0
       0                    7800       0   29.25
Permanent Ineff=
       F       T
#Block Obstruct= 2 ,-1
    7555    7800   28.59    8785    9150    28.5
Bank Sta=4912.3,5074.92
XS Rating Curve= 0 ,0
Exp/Cntr=0.3,0.1

Type RM Length L Ch R = 1 ,12968.9 ,17.39,106.91,216.28
BEGIN DESCRIPTION:
Added cross-section is interpolated in channel banks and uses 2001 LiDAR in the overbanks and survey in the project boundary
Watearth, 2018
END DESCRIPTION:
XS GIS Cut Line= 6
  3180979.16700113780760.9905898 3180479.514130213780248.0903548
 3179996.729097313779845.2121239 3179882.952173413779738.8971702
 3178730.283610413778736.3001258 3176207.777386113775942.0164816
#Sta/Elev= 30
 3555.79   30.06 3739.77   30.04 3769.61   38.35 3794.47   39.65 4082.88   29.48
 4301.47   31.08 4464.49   25.92 4513.89   29.42 4796.27   30.52 4912.71   26.34
 4933.87   12.31 4993.81   11.62 5034.35   13.12 5075.33   26.39 5231.73   30.19
 6090.03   25.85 6679.04   30.85 7303.27   26.88 7353.21    31.5    7517   29.05
 7552.81    17.5 7704.47    17.5 7752.46   29.25    8730    28.5 8757.05    19.5
    9256    19.5    9292    28.5 9457.99    32.310273.53   28.08 10348.6   28.16
#Mann= 9 ,-1 , 0
 3555.79     .07       0 4912.71    .015       0 5075.33     .07       0
 6679.04     .12       0    7517    .012       0 7752.46     .12       0
    8730    .012       0    9292     .12       010273.53     .07       0
#XS Ineff= 2 , 0
       0                 7752.46       0   29.25
Permanent Ineff=
       F       T
#Block Obstruct= 2 ,-1
    7517 7752.46   29.05    8730    9292    28.5
Bank Sta=4912.71,5075.33
XS Rating Curve= 0 ,0
Exp/Cntr=0.3,0.1

Type RM Length L Ch R = 1 ,12861.99,23.46,20.49,20.23
BEGIN DESCRIPTION:
Dixie Farm Road
END DESCRIPTION:
XS GIS Cut Line= 6
      3180986.03    13780756.525     3180212.405    13779942.422
     3180054.062    13779766.104     3179951.523    13779640.191
     3179802.986    13779482.528 3176685.203422213775994.0439423
#Sta/Elev= 30
 3563.07 30.43433657.906 32.84263752.742 30.28683792.673 42.79344162.034 29.7841
4311.775 31.2691 4511.43 26.03554581.309 29.73314819.431 29.3932 4918.69   26.34
 4939.85   12.31 4999.79   11.45 5040.33   13.12 5081.31   26.395208.568 29.2396
5561.795 28.33466111.139 25.92756610.542 27.40086975.106 32.3665 7214.82 31.0888
7274.749 27.82187409.587 31.7866 7439.54 28.45547472.406    17.57831.415    17.5
7831.435   29.257853.396 31.6406 8960.03   29.18 9905.07 31.79939980.79428.61994
#Mann= 6 ,-1 , 0
 3563.07     .07       0 4918.69    .015       0 5081.31     .07       0
5561.795     .12       0 7439.54    .012       07831.435     .12       0
#XS Ineff= 1 ,-1
 4092.84 4318.79   31.13
Permanent Ineff=
       F
#Block Obstruct= 3 ,-1
 3462.38 3820.91   40.53 4096.74  4636.3   29.75 7439.54 7831.44 28.4554
Bank Sta=4918.69,5081.31
XS Rating Curve= 0 ,0
Exp/Cntr=0.5,0.3

Type RM Length L Ch R = 1 ,12841.5 ,137.38,122.01,125.78
BEGIN DESCRIPTION:
Dixie Farm Road
END DESCRIPTION:
XS GIS Cut Line= 6
      3181000.53    13780742.748     3180227.097    13779928.849
     3180069.265      13779753.1     3179966.575    13779627.002
     3179817.723    13779469.004     3177053.142    13776375.862
#Sta/Elev= 30
 3560.57      31 3664.54   33.17  3751.5   31.11  3762.2   31.95 3807.84   42.45
 3820.36    42.6 4001.02   40.11 4223.52   30.46 4339.44    31.1  4535.4   28.64
 4680.06   30.18 4907.75   27.86 4923.69   26.34 4944.85   12.31 4959.51   14.16
 5004.79   11.45 5045.33   13.12 5086.31   26.39 5104.36   28.23 5190.73   29.66
 5312.42    26.8 5574.02   26.38 5867.26    27.9 6060.62   27.45 6101.34   25.75
 6335.54    28.1 6536.72   27.79 6575.62   26.17 6874.96   27.23 9447.81   27.42
#Mann= 5 ,-1 , 0
 3560.57     .07       0 4923.69    .015       0 5086.31     .07       0
 5574.02     .12       0 6874.96     .07       0
#XS Ineff= 2 , 0
       0    4915    28.5    5093       0    28.5
Permanent Ineff=
       F       F
#Block Obstruct= 2 ,-1
  3522.7 3819.65    42.6 4374.81 4629.06   29.75
Bank Sta=4923.69,5086.31
XS Rating Curve= 0 ,0
Exp/Cntr=0.5,0.3

Type RM Length L Ch R = 3 ,12780   ,,,
BEGIN DESCRIPTION:
Bridge at Dixie Farm Road
END DESCRIPTION:
Bridge Culvert--1,0,-1,-1, 0
Deck Dist Width WeirC Skew NumUp NumDn MinLoCord MaxHiCord MaxSubmerge Is_Ogee
8,70,2.6,0, 11, 11, , , 0.95, 0, 0,0,,
    3743    3838    3993    4208    4427    4905    4905    5095    5095    6787
    9645
   31.56   47.55   43.28   34.08   30.67   29.64   30.45   30.45   29.96   28.73
   28.93
       0       0       0       0       0       0   26.87   26.87       0       0
       0
    3743    3838    3993    4208    4427    4905    4905    5095    5095    6787
    9645
   31.56   47.55   43.28   34.08   30.67   29.64   30.45   30.45   29.96   28.73
   28.93
       0       0       0       0       0       0   26.87   26.87       0       0
       0
Pier Skew, UpSta & Num, DnSta & Num=  ,4973, 4 ,4973, 4 , 3 , 3 , 0 ,,
    1.35    1.35    2.75    2.75
       0   24.12   24.12      27
    1.35    1.35    2.75    2.75
       0   24.12   24.12      27
Pier Skew, UpSta & Num, DnSta & Num=  ,5027, 4 ,5027, 4 , 3 , 3 , 0 ,,
    1.35    1.35    2.75    2.75
       0   24.12   24.12      27
    1.35    1.35    2.75    2.75
       0   24.12   24.12      27
BR Coef=-1 , 1 , 0 ,, 0 ,,,0.8,-1,2,0,
WSPro=,,,, 1 ,,,, 0 ,,,, 0 ,,,,-1 ,-1 ,-1 , 0 , 0 , 0 , 0 , 0
BC Design=,, 0 ,, 0 ,,,,,,
BC HTab HWMax=42.6
BC Use User HTab Curves=0
BC User HTab FreeFlow(D)= 0

Type RM Length L Ch R = 1 ,12719.49,82.03,80.03,78.7
BEGIN DESCRIPTION:
Dixie Farm Road
END DESCRIPTION:
XS GIS Cut Line= 6
      3181087.52    13780660.085     3180160.483    13779675.077
     3178861.536    13778199.463     3178595.745    13777832.907
     3178310.205    13777506.576     3177175.897    13776281.795
#Sta/Elev= 30
  3569.2   33.85 3578.98   31.25 3674.47   33.22 3759.35    31.5 3802.92   41.24
 4138.55   32.21 4257.87   33.29 4305.34   30.13 4713.78   29.39 4805.67   26.95
    4894    29.1 4918.69   26.34 4939.85   12.31 4954.51   14.16 4999.79   11.45
 5040.33   13.12 5081.31   26.39 5099.36   28.23 5682.28   25.67 6089.81   25.42
 6180.46   27.47 7073.21   25.43 7141.65   27.21 7461.64   26.35 7497.41   28.51
 7522.44   26.41  8053.9   26.21 9175.42   27.67 9367.14   30.46 9445.16   28.21
#Mann= 3 ,-1 , 0
  3569.2     .07       0 4918.69    .015       0 5081.31     .07       0
#XS Ineff= 2 , 0
       0    4910    28.5    5088       0    28.5
Permanent Ineff=
       F       F
#Block Obstruct= 1 ,-1
 3431.66 3800.16   41.26
Bank Sta=4918.69,5081.31
XS Rating Curve= 0 ,0
Exp/Cntr=0.5,0.3

Type RM Length L Ch R = 1 ,12639.46,416.4,490.53,601.75
BEGIN DESCRIPTION:
Dixie Farm Road
END DESCRIPTION:
XS GIS Cut Line= 6
      3181145.51    13780604.976     3180374.017     13779793.12
     3180221.296    13779623.061     3180117.097    13779495.111
     3179965.095    13779333.769     3177228.583    13776247.774
#Sta/Elev= 30
 3579.01   31.39 3683.02    33.4 3837.34    30.4 4010.12   31.74 4267.18   29.52
 4316.46   32.08 4461.42   27.89  4624.3   29.51 4848.91   28.62 4918.69   26.34
 4939.85   12.31 4954.51   14.16 4999.79   11.45 5040.33   13.12 5081.31   26.39
 5099.36   28.23 5449.44   28.71 5718.26   26.42 5962.74   27.02 6120.42   24.49
  6190.8   27.08 6771.26   28.71  7475.4   26.69 7497.76   28.59 7529.64    26.3
 8232.98   28.96 8934.72   29.22 9078.74   26.98 9146.06   28.61 9438.76   28.32
#Mann= 3 ,-1 , 0
 3579.01     .07       0 4918.69     .03       0 5081.31     .07       0
#XS Ineff= 1 ,-1
    4400    4560    29.5
Permanent Ineff=
       F
#Block Obstruct= 3 ,-1
 3522.12 3683.46    33.4 3726.16 4315.45    31.8 5970.42 6241.18      24
Bank Sta=4918.69,5081.31
XS Rating Curve= 0 ,0
Exp/Cntr=0.3,0.1

Type RM Length L Ch R = 1 ,12148.93,15.56,15.01,15.44
BEGIN DESCRIPTION:
Pipe
END DESCRIPTION:
XS GIS Cut Line= 6
       3181355.9    13780401.899     3180636.389    13779385.689
     3180607.489    13779334.047     3180496.544    13779158.394
     3179643.004    13777981.895     3177645.056    13775527.302
#Sta/Elev= 30
 3645.16   30.19 3691.71   32.91 3761.08   33.55 3944.78   29.22 4078.61   28.91
 4151.67    31.2 4224.38   28.69 4451.58   30.69 4886.12   29.53 4911.11   27.31
 4919.12   26.85    4950   16.91 5005.51   12.17 5040.84   13.37 5065.55   22.71
 5087.75   27.13 5819.34   27.95 5948.28   26.48 5982.72    23.3 6042.23   26.51
 6301.16   28.23 7550.85   26.32 8439.94   28.47 8863.08   27.45 8942.56   28.87
 8988.31   27.38 9096.58    28.1 9143.65   25.75 9192.97   27.67 9775.68   27.92
#Mann= 3 ,-1 , 0
 3645.16     .07       0 4911.11     .03       0 5087.75     .07       0
#XS Ineff= 3 ,-1
    4408 4911.11   27.31 4172.21 4407.77   30.43 5087.75 9775.68   27.13
Permanent Ineff=
       F       F       F
#Block Obstruct= 3 ,-1
 3563.88 3759.44   33.55 3768.01 4157.28   31.16    5843 6145.62      24
Bank Sta=4911.11,5087.75
XS Rating Curve= 0 ,0
Exp/Cntr=0.3,0.1

Type RM Length L Ch R = 3 ,12140   ,,,
BEGIN DESCRIPTION:
Pipe Crossing downstream of Dixie Farm Road
END DESCRIPTION:
Bridge Culvert--1,0,-1,-1, 0
Deck Dist Width WeirC Skew NumUp NumDn MinLoCord MaxHiCord MaxSubmerge Is_Ogee
4,5,2.6,0, 4, 4, , , 0.95, 0, 0,0,,
    4915    4935    5065    5085
      27   30.28   30.28    26.5
      26   29.28   29.28    25.5
    4915    4935    5065    5085
      27   30.28   30.28    26.5
      26   29.28   29.28    25.5
Pier Skew, UpSta & Num, DnSta & Num=  ,4940, 4 ,4940, 4 , 3 , 3 , 0 ,,
    1.15    1.15       2       2
       0   27.28   27.28      30
    1.15    1.15       2       2
       0   27.28   27.28      30
Pier Skew, UpSta & Num, DnSta & Num=  ,4980, 4 ,4980, 4 , 3 , 3 , 0 ,,
    1.15    1.15       2       2
       0   27.28   27.28      30
    1.15    1.15       2       2
       0   27.28   27.28      30
Pier Skew, UpSta & Num, DnSta & Num=  ,5020, 4 ,5020, 4 , 3 , 3 , 0 ,,
    1.15    1.15       2       2
       0   27.28   27.28      30
    1.15    1.15       2       2
       0   27.28   27.28      30
Pier Skew, UpSta & Num, DnSta & Num=  ,5060, 4 ,5060, 4 , 3 , 3 , 0 ,,
    1.15    1.15       2       2
       0   27.28   27.28      30
    1.15    1.15       2       2
       0   27.28   27.28      30
BR Coef=-1 , 1 , 0 ,, 0 ,,,0.8,-1,2,0,
WSPro=,,,, 1 ,,,, 0 ,,,, 0 ,,,,-1 ,-1 ,-1 , 0 , 0 , 0 , 0 , 0
BC Design=,, 0 ,, 0 ,,,,,,
BC HTab HWMax=33.55
BC Use User HTab Curves=0
BC User HTab FreeFlow(D)= 0

Type RM Length L Ch R = 1 ,12133.92,783.2,856.57,758.1
BEGIN DESCRIPTION:
Pipe
END DESCRIPTION:
XS GIS Cut Line= 6
      3181368.14    13780393.231     3180649.091     13779377.67
     3180620.391    13779326.387     3180508.961    13779149.965
     3179654.904    13777972.755     3177658.226    13775517.257
#Sta/Elev= 30
 3648.12   29.99 3696.59   32.85 3770.37   33.51 3837.77   30.71 4009.58   29.08
 4149.44   31.21 4218.99   28.69  4477.4   30.68 4891.01   29.55 4915.77   27.36
  4923.1   26.61    4950   16.91 5005.51   12.17 5040.84   13.37    5050   17.67
 5089.64   27.11 5827.87   27.92 5949.91   26.36  5987.9   22.86 6035.52   26.28
 6293.55   28.15 7554.56   26.34 7604.89   27.68 8865.52   27.41 8953.17   28.71
  9001.9   27.27 9099.26   28.28 9148.63   25.72 9193.65   27.64 9779.13   27.71
#Mann= 3 ,-1 , 0
 3648.12     .07       0 4915.77     .03       0 5089.64     .07       0
#XS Ineff= 3 ,-1
    4356 4915.77   27.36 4164.23 4355.23    30.5 5089.64 9779.13   27.11
Permanent Ineff=
       F       F       F
#Block Obstruct= 3 ,-1
 3594.59 3770.59   33.52 3780.32 4151.45   31.13 5866.89 6169.51      24
Bank Sta=4915.77,5089.64
XS Rating Curve= 0 ,0
Exp/Cntr=0.3,0.1

Type RM Length L Ch R = 1 ,11277.35,10.27,10,12.95
BEGIN DESCRIPTION:
access road
END DESCRIPTION:
XS GIS Cut Line= 5
       3181893.6    13779902.011     3181126.859    13778667.748
     3180984.568    13778501.444     3180920.084    13778438.803
     3177890.011    13775324.954
#Sta/Elev= 30
 3439.76    28.7 3489.05   33.33  3580.2   32.36 3612.87   28.76 3634.66   30.47
 3713.38   31.47 4796.46   27.93 4840.61   26.46 4954.32   15.67 4968.63   12.07
 4998.17   10.97 5026.06    13.5  5032.5   16.16 5074.39   21.29 5187.96   28.27
 6113.06   25.27 6143.62   23.13 6260.94   26.34 7271.38   27.47 7305.37   26.01
 7589.29   26.94 7686.42   29.02 7756.05   26.92 8225.92   26.61 8643.39    28.7
 8715.62   27.08 8872.32   27.51 8917.04   25.94 9052.72   27.64 9546.37   27.96
#Mann= 3 ,-1 , 0
 3439.76     .07       0 4796.46     .03       0 5187.96     .07       0
#XS Ineff= 1 ,-1
 3552.26 4430.19    30.1
Permanent Ineff=
       F
#Block Obstruct= 3 ,-1
 3374.08 3488.52   33.32 3576.75 3637.63    29.7 6097.84 6265.07      24
Bank Sta=4796.46,5187.96
XS Rating Curve= 0 ,0
Exp/Cntr=0.5,0.3

Type RM Length L Ch R = 1 ,11267.35,51.35,50.03,65.33
BEGIN DESCRIPTION:
access road
END DESCRIPTION:
XS GIS Cut Line= 5
      3181902.09    13779896.734     3181134.952    13778661.825
     3180991.866    13778494.593     3180927.152    13778431.729
     3177896.965    13775317.761
#Sta/Elev= 30
 3436.08   28.53 3492.11   33.37 3582.05   32.35 3614.73   28.71 3636.51   30.49
  3714.3   31.45 4796.46   27.93 4840.61   26.46 4954.32   15.67 4968.63    11.4
 4998.17   10.97 5017.01    11.6  5032.5   16.16 5074.39   21.29 5202.44    28.1
 6116.88   25.27 6147.95   22.99 6256.81   26.22  7270.8   27.46 7305.64      26
 7573.53   26.97 7684.92   29.04 7750.79    26.9 8225.11    26.6  8644.3   28.68
 8721.75   27.03 8873.03   27.51 8918.19   25.92 9066.97   27.65 9545.16   27.97
#Mann= 3 ,-1 , 0
 3436.08     .07       0 4796.46     .03       0 5202.44     .07       0
#XS Ineff= 4 ,-1
    4441    4965    15.1  3512.2 3728.46   30.66    5015 9545.16    15.1
    4250    4440   30.05
Permanent Ineff=
       F       F       F       F
#Block Obstruct= 3 ,-1
  3377.2 3491.25   33.36 3582.16 3641.54   29.72 6097.84 6312.86      24
Bank Sta=4796.46,5202.44
XS Rating Curve= 0 ,0
Exp/Cntr=0.5,0.3

Type RM Length L Ch R = 2 ,11242   ,,,
BEGIN DESCRIPTION:
Culverts at access road
END DESCRIPTION:
Bridge Culvert--1,0,-1,-1, 0
Deck Dist Width WeirC Skew NumUp NumDn MinLoCord MaxHiCord MaxSubmerge Is_Ogee
5,31,2.6,0, 14, 14, , , 0.95, 0, 0,0,,
    4420    4674    4806    4852    4894    4938    4979    5026    5037    5081
    5128    5174    5300    5700
    29.8   28.62   27.91   26.11   21.58   17.72   16.12   16.67   17.66   21.07
    24.7   27.54   27.05   25.86
       0       0       0       0       0       0       0       0       0       0
       0       0       0       0
    4420    4674    4806    4852    4894    4938    4979    5026    5037    5081
    5128    5174    5300    5700
    29.8   28.62   27.91   26.11   21.58   17.72   16.12   16.67   17.66   21.07
    24.7   27.54   27.05   25.86
       0       0       0       0       0       0       0       0       0       0
       0       0       0       0
Multiple Barrel Culv=2,3,6,31,0.012,0.5,1,10,1,11.51,11.04, 6,Culvert #1  , 0 ,5
  4972.5  4972.5  4979.5  4979.5  4986.5  4986.5  4993.5  4993.5  5000.5  5000.5
  5007.5  5007.5
Culvert Bottom n=0.012
BC Design=,, 0 ,, 0 ,,,,,,
BC HTab HWMax=33.37
BC Use User HTab Curves=0
BC User HTab FreeFlow(D)= 0

Type RM Length L Ch R = 1 ,11217.32,41.08,40.25,50.1
BEGIN DESCRIPTION:
access road
END DESCRIPTION:
XS GIS Cut Line= 5
      3181944.56     13779870.35     3181175.417     13778632.21
     3181028.359    13778460.335     3180962.497    13778396.355
     3177937.694    13775285.038
#Sta/Elev= 30
 3428.46   28.46  3518.1   33.53    3583   32.37 3616.92   28.52 3710.54   31.35
 4796.46   27.93 4840.61   26.46 4937.86   17.48 4963.88   13.81 4968.63   10.98
 4998.17   10.97 5017.01   10.97  5032.5   16.16 5074.39   21.29 5184.62   27.32
  5876.9   26.63 6090.28   25.05 6161.38   22.29 6283.94   26.25 6653.24   27.43
  7259.3   27.42 7303.22   25.97 7668.72   29.16 7725.02   26.84 8457.34   26.79
 8638.36   28.49 8868.08   27.53 8918.98   25.55 9132.18   27.73  9543.4   28.08
#Mann= 3 ,-1 , 0
 3428.46     .07       0 4796.46     .03       0 5184.62     .07       0
#XS Ineff= 3 ,-1
    3729    4965    15.1 3523.58 3728.46    30.6    5015  9543.4    15.1
Permanent Ineff=
       F       F       F
#Block Obstruct= 3 ,-1
 3350.62  3516.8    33.5 3586.04 3644.39    29.7 6058.06 6368.36      24
Bank Sta=4796.46,5184.62
XS Rating Curve= 0 ,0
Exp/Cntr=0.5,0.3

Type RM Length L Ch R = 1 ,11177.08,1710.95,1323.5,800.41
BEGIN DESCRIPTION:
access road
END DESCRIPTION:
XS GIS Cut Line= 5
      3181978.54    13779849.243     3181207.789    13778608.517
     3181057.553    13778432.928     3180990.772    13778368.057
     3177962.527    13775260.182
#Sta/Elev= 30
 3423.05   29.61 3441.22   27.89 3482.82   32.52 3534.26   33.55 3584.66   32.47
 3622.74   28.47 3710.36   31.28  4795.6   28.07 4925.61   21.29  4967.5   16.16
 4973.94    13.5 5001.83   10.97 5031.37   12.07 5045.68   15.67 5159.39   26.46
 5203.54   27.93 5699.66   25.97 6013.02   26.92 6240.68   22.53 6321.14   26.33
 6684.56   27.51 7253.62    27.4 7304.26   25.95 7684.82      29 7753.38   27.03
 8246.86   26.57 8636.02   28.34 8866.92   27.52 8922.34   25.29 9547.14   28.77
#Mann= 3 ,-1 , 0
 3423.05     .07       0  4795.6     .03       0 5203.54     .07       0
#XS Ineff= 1 ,-1
    3525    3725    30.5
Permanent Ineff=
       F
#Block Obstruct= 3 ,-1
 3322.52 3534.57   33.54 3591.05 3654.43    29.7 6099.25 6323.21      24
Bank Sta=4795.6,5203.54
XS Rating Curve= 0 ,0
Exp/Cntr=0.3,0.1

Type RM Length L Ch R = 1 ,9853.579,20.09,20.6,21.08
BEGIN DESCRIPTION:
Pipe
END DESCRIPTION:
XS GIS Cut Line= 6
      3183471.69    13778048.058      3181849.41    13777419.695
     3181743.585    13777377.789     3181547.757    13777280.122
     3180155.501    13776757.205     3178103.947    13774794.824
#Sta/Elev= 30
    3202   29.25 3241.52   29.51 3288.48   32.28 3380.99    31.9 3427.36   28.73
 4145.11   29.05 4778.32   26.53 4943.09   26.94 4980.26   22.54 5001.58   17.37
 5007.28   13.58 5015.98   14.21 5056.91    25.3  5091.3   27.54  5133.3   25.79
 5229.19   26.12  5358.1   27.22 5980.64    25.5 6136.15   26.01 6182.74   20.77
 6241.97   25.32 6356.37   26.96 7011.36   27.19 7164.92    24.9 7227.94   26.55
 7621.64   27.08 8605.39    27.2 8711.48   25.64 8880.53   27.65 9600.58   27.61
#Mann= 7 ,-1 , 0
    3202     .07       0 4778.32     .12       0 4943.09     .03       0
 5056.91     .12       0 5229.19     .07       0 5980.64     .12       0
 6356.37     .07       0
#XS Ineff= 2 , 0
         4904.56   25.77 5103.47           25.31
Permanent Ineff=
       F       F
#Block Obstruct= 3 ,-1
  3087.6 3302.62   32.15                         6120.77 6249.95      24
Bank Sta=4943.09,5056.91
XS Rating Curve= 0 ,0
Exp/Cntr=0.3,0.1

Type RM Length L Ch R = 3 ,9843    ,,,
BEGIN DESCRIPTION:
Pipe crossing
END DESCRIPTION:
Bridge Culvert--1,0,-1,-1, 0
Deck Dist Width WeirC Skew NumUp NumDn MinLoCord MaxHiCord MaxSubmerge Is_Ogee
5,10,2.6,0, 6, 6, , , 0.95, 0, 0,0,,
    4905    4909    4909    5111    5111    5115
   31.85   31.85   31.85   31.85   31.85   31.85
       0       0   27.77   27.77       0       0
    4905    4909    4909    5111    5111    5115
   31.85   31.85   31.85   31.85   31.85   31.85
       0       0   27.77   27.77       0       0
Pier Skew, UpSta & Num, DnSta & Num=  ,5000, 4 ,5000, 4 , 3 , 3 , 0 ,,
    1.15    1.15       2       2
       0   25.77   25.77      28
    1.15    1.15       2       2
       0   25.77   25.77      28
BR Coef=-1 , 1 , 0 ,, 0 ,,,0.8,-1,2,0,
WSPro=,,,, 1 ,,,, 0 ,,,, 0 ,,,,-1 ,-1 ,-1 , 0 , 0 , 0 , 0 , 0
BC Design=,, 0 ,, 0 ,,,,,,
BC HTab HWMax=32.28
BC Use User HTab Curves=0
BC User HTab FreeFlow(D)= 0

Type RM Length L Ch R = 1 ,9832.981,1692.79,1291.58,208.05
BEGIN DESCRIPTION:
Pipe
END DESCRIPTION:
XS GIS Cut Line= 6
      3183478.92    13778029.411     3181856.635    13777401.045
     3181751.745    13777359.509     3181555.758    13777261.763
     3180166.367    13776739.922     3178118.151    13774780.813
#Sta/Elev= 30
 3198.01   29.32  3230.4   29.55 3283.94   32.35 3370.12   31.99 3415.88   28.84
 4131.76   29.07    4778   26.37 4943.09   26.94 4980.26   22.54 5001.58   17.37
 5007.28   13.58 5015.98   14.21 5019.37   16.15 5056.91    25.3  5088.4   27.11
  5173.2   25.35 5229.54   26.57 6030.46   25.97 6117.24    26.2 6171.22    20.3
 6208.16   24.24 6365.52   27.04 6986.74   27.21 7165.68   24.86 7226.76   26.53
 7590.12   27.02  8588.7   27.17 8702.08   25.67 8879.34   27.53 9588.03   27.97
#Mann= 7 ,-1 , 0
 3198.01     .07       0    4778     .12       0 4943.09     .03       0
 5056.91     .12       0 5229.54     .07       0 6030.46     .12       0
 6365.52     .07       0
#XS Ineff= 2 , 0
         4912.59   25.74  5097.4           25.32
Permanent Ineff=
       F       F
#Block Obstruct= 3 ,-1
 3071.67 3294.65   32.25                         6087.27 6257.57      24
Bank Sta=4943.09,5056.91
XS Rating Curve= 0 ,0
Exp/Cntr=0.3,0.1

Type RM Length L Ch R = 1 ,8541.402,21.05,20.65,40.76
BEGIN DESCRIPTION:
access road
END DESCRIPTION:
XS GIS Cut Line= 6
      3185305.62    13775821.809     3183495.582    13775258.174
      3182272.49    13776150.358     3181785.978    13776520.468
     3180328.925    13776624.809     3178210.956    13774693.324
#Sta/Elev= 30
 1372.66   31.55 1528.41   35.26 1640.56   32.06 2347.11   33.87 3530.74   31.13
 3572.03    32.5 3809.46   30.62  3841.6   32.03  4385.2   26.21 4591.91   26.51
 4765.45   22.67  4893.7    20.9 4926.39   23.82 4972.96   21.19  4988.4   15.31
 5002.65   13.66 5027.04   21.86 5039.34   23.95 5088.56   25.29 5377.32   25.45
 5717.56   26.67 6091.16   24.98 6265.05   24.54 6309.84   19.46 6366.65   24.57
 6499.07   26.52 6971.55   26.91 7411.92   24.58 7454.71   26.35 9720.97   28.65
#Mann= 7 ,-1 , 0
 1372.66     .07       0 4765.45     .12       0 4972.96     .03       0
 5027.04     .12       0 5377.32     .07       0 6091.16     .12       0
 6499.07     .07       0
#Block Obstruct= 1 ,-1
 6264.84 6408.49      24
Bank Sta=4972.96,5027.04
XS Rating Curve= 0 ,0
Exp/Cntr=0.5,0.3

Type RM Length L Ch R = 1 ,8520.751,45.81,40.9,33.73
BEGIN DESCRIPTION:
access road
END DESCRIPTION:
XS GIS Cut Line= 6
      3185481.51    13773783.958     3182260.512     13776134.34
     3182074.249    13776272.396     3181812.063     13776475.75
     3180353.338    13776582.446     3178246.335    13774663.373
#Sta/Elev= 30
  807.47   34.12  987.02   35.47 2772.48    33.6 3196.28   31.39 3843.46   32.07
 4761.74   24.24 4798.82   23.17  4821.5   26.06 4853.33   26.31 4926.39   23.82
 4972.96   21.19  4988.4   15.31 5002.65   13.66 5027.04   21.86 5039.34   23.95
 5384.18   25.72 6079.78   24.78    6186   24.56 6237.04   19.29  6289.1   24.97
 6334.14   23.46 6573.32   27.46 7390.78   24.51 7446.44   26.33 8757.34   25.52
 9073.34    28.6 9162.56   27.43 9228.52   29.42 9317.62   27.74 9671.17      28
#Mann= 7 ,-1 , 0
  807.47     .07       0 4761.74     .12       0 4926.39     .03       0
 5039.34     .12       0 5384.18     .07       0 6079.78     .12       0
 6573.32     .07       0
#XS Ineff= 2 , 0
       0    4905      28    5095       0      28
Permanent Ineff=
       F       F
#Block Obstruct= 1 ,-1
 6185.62 6282.46      24
Bank Sta=4926.39,5039.34
XS Rating Curve= 0 ,0
Exp/Cntr=0.5,0.3

Type RM Length L Ch R = 3 ,8500    ,,,
BEGIN DESCRIPTION:
Bridge at access road
END DESCRIPTION:
Bridge Culvert--1,0,-1,-1, 0
Deck Dist Width WeirC Skew NumUp NumDn MinLoCord MaxHiCord MaxSubmerge Is_Ogee
5,20,2.6,0, 15, 15, , , 0.95, 0, 0,0,,
     910    4365    4765    4830    4910    4910    4949    5000    5090    5090
    5141    5192    5239    5409    6050
   35.12   27.51   26.43   27.43   28.47    29.4    29.4    29.4    29.4   28.46
   28.14   27.16   26.31   25.64   26.78
       0       0       0       0       0   27.05   27.05   27.05   27.05       0
       0       0       0       0       0
     910    4365    4765    4830    4910    4910    4949    5000    5090    5090
    5141    5192    5239    5409    6050
   35.12   27.51   26.43   27.43   28.47    29.4    29.4    29.4    29.4   28.46
   28.14   27.16   26.31   25.64   26.78
       0       0       0       0       0   27.05   27.05   27.05   27.05       0
       0       0       0       0       0
Pier Skew, UpSta & Num, DnSta & Num=  ,4983, 4 ,4983, 4 , 3 , 3 , 0 ,,
    1.35    1.35    2.35    2.35
       0    24.7    24.7      28
    1.35    1.35    2.35    2.35
       0    24.7    24.7      28
Pier Skew, UpSta & Num, DnSta & Num=  ,5017, 4 ,5017, 4 , 3 , 3 , 0 ,,
    1.35    1.35    2.35    2.35
       0    24.7    24.7      28
    1.35    1.35    2.35    2.35
       0    24.7    24.7      28
BR Coef=-1 , 1 , 0 ,, 0 ,,,0.8,0,2,0,
WSPro=,,,, 1 ,,,, 0 ,,,, 0 ,,,,-1 ,-1 ,-1 , 0 , 0 , 0 , 0 , 0
BC Design=,, 0 ,, 0 ,,,,,,
BC HTab HWMax=35.47
BC Use User HTab Curves=0
BC User HTab FreeFlow(D)= 0

Type RM Length L Ch R = 1 ,8479.856,223.22,113.87,115.41
BEGIN DESCRIPTION:
access road
END DESCRIPTION:
XS GIS Cut Line= 6
      3185443.18    13773709.313     3182095.966    13776209.823
     3182050.794    13776239.959     3181800.884    13776427.306
     3180374.325    13776547.457     3178274.555    13774634.972
#Sta/Elev= 30
  798.92   34.85 2330.47   34.39 3457.24   30.93 3865.03   31.87 4467.25   25.51
 4677.21   26.54 4737.57   23.88 4824.17   24.61 4972.96   21.19  4988.4   15.31
 5002.65   13.66 5027.04   21.86 5039.34   23.95 5088.56    24.6 5343.18   25.37
 5658.15   26.55 6049.71   24.78  6126.5   24.53 6199.71   18.83 6282.23   25.45
 6323.54   24.36 6453.44   26.42 6866.78   26.79 7355.41   24.22 7408.31   26.25
 8561.06   26.72  8665.4   26.31 8697.47   24.47 8754.96   27.06 9615.46   28.27
#Mann= 7 ,-1 , 0
  798.92     .07       0 4737.57     .12       0 4972.96     .03       0
 5027.04     .12       0 5343.18     .07       0 6049.71     .12       0
 6453.44     .07       0
#XS Ineff= 2 , 0
       0    4905      28    5095       0      28
Permanent Ineff=
       F       F
#Block Obstruct= 1 ,-1
 6126.29 6288.97      24
Bank Sta=4972.96,5027.04
XS Rating Curve= 0 ,0
Exp/Cntr=0.5,0.3

Type RM Length L Ch R = 1 ,8365.985,16.87,15.11,13.12
BEGIN DESCRIPTION:
Pipe
END DESCRIPTION:
XS GIS Cut Line= 6
      3185321.51    13773582.005      3182368.95    13775744.972
     3182036.313    13776106.021     3181831.127     13776312.12
     3180321.163    13776436.293     3178306.549    13774607.959
#Sta/Elev= 30
  808.79    33.6 1265.93   36.33 2146.41    35.1 3103.19   31.17 3700.86   32.53
  4409.7   30.33 4449.07    27.2 4958.67   23.85 4978.62   19.92 4996.71   13.82
 5007.32   13.09 5041.33    24.3 5310.15   25.48  5810.4   26.23 6028.52   24.56
  6067.1   22.02 6108.82   23.16  6139.7   18.48 6202.02   24.98  6410.7   25.53
  7177.4   25.79  7249.8    23.8 7421.74   25.52 7442.25   27.72 7474.83   25.53
 8444.79    26.8 8566.46    25.2 8621.69   27.15 8810.02   27.95 9486.25   28.91
#Mann= 7 ,-1 , 0
  808.79     .07       0  4409.7     .12       0 4958.67     .03       0
 5041.33     .12       0 5310.15     .07       0  5810.4     .12       0
  6410.7     .07       0
#XS Ineff= 2 , 0
       0 4958.67   23.85 5041.33       0    24.3
Permanent Ineff=
       F       F
#Block Obstruct= 2 ,-1
 6025.08 6240.73      24 9279.07 9430.98   28.51
Bank Sta=4958.67,5041.33
XS Rating Curve= 0 ,0
Exp/Cntr=0.3,0.1

Type RM Length L Ch R = 3 ,8358    ,,,
BEGIN DESCRIPTION:
Pipe crossing
END DESCRIPTION:
Bridge Culvert--1,0,-1,-1, 0
Deck Dist Width WeirC Skew NumUp NumDn MinLoCord MaxHiCord MaxSubmerge Is_Ogee
3,10,2.6,0, 6, 6, , , 0.95, 0, 0,0,,
  4912.5  4915.5  4915.5  5084.5  5084.5  5087.5
   29.55   29.55   29.55   29.55   29.55   29.55
       0       0   26.55   26.55       0       0
  4912.5  4915.5  4915.5  5084.5  5084.5  5087.5
   29.55   29.55   29.55   29.55   29.55   29.55
       0       0   26.55   26.55       0       0
Pier Skew, UpSta & Num, DnSta & Num=  ,4979, 4 ,4979, 4 , 3 , 3 , 0 ,,
    1.15    1.15       2       2
       0   24.55   24.55      27
    1.15    1.15       2       2
       0   24.55   24.55      27
Pier Skew, UpSta & Num, DnSta & Num=  ,5021, 4 ,5021, 4 , 3 , 3 , 0 ,,
    1.15    1.15       2       2
       0   24.55   24.55      27
    1.15    1.15       2       2
       0   24.55   24.55      27
BR Coef=-1 , 1 , 0 ,, 0 ,,,0.8,-1,2,0,
WSPro=,,,, 1 ,,,, 0 ,,,, 0 ,,,,-1 ,-1 ,-1 , 0 , 0 , 0 , 0 , 0
BC Design=,, 0 ,, 0 ,,,,,,
BC HTab HWMax=36.33
BC Use User HTab Curves=0
BC User HTab FreeFlow(D)= 0

Type RM Length L Ch R = 1 ,8350.878,1425.46,2104.01,879.43
BEGIN DESCRIPTION:
Pipe
END DESCRIPTION:
XS GIS Cut Line= 6
      3185312.64    13773569.904     3182358.896    13775733.743
     3182025.374    13776095.757     3181821.248    13776300.795
     3180338.461    13776421.718     3178320.664    13774597.222
#Sta/Elev= 30
  804.18   33.53  1267.3   36.28 1523.12   34.52 2135.96   35.09 3084.62   31.23
  3673.4   32.51  4396.1   30.62 4444.68   27.29 4958.67   23.85 4978.62   19.92
 4996.71   13.82 5007.32   13.09 5041.33    24.3 5312.48   25.66 5811.38   26.13
  6000.7   24.63  6045.1   20.81  6094.1   20.13 6106.62   22.48 6141.98   21.64
 6187.38   25.06 6461.72   25.48 7128.54    25.8 7233.08   23.64 7401.96   26.65
 8421.08   26.84 8533.28   24.63 8592.38    27.2 8791.64   28.22 9455.35    28.9
#Mann= 7 ,-1 , 0
  804.18     .07       0  4396.1     .12       0 4958.67     .03       0
 5041.33     .12       0 5312.48     .07       0 5811.38     .12       0
 6461.72     .07       0
#XS Ineff= 2 , 0
       0 4958.67   23.85 5041.33       0    24.3
Permanent Ineff=
       F       F
#Block Obstruct= 2 ,-1
 5999.64 6314.64      24  9255.1 9426.15   28.51
Bank Sta=4958.67,5041.33
XS Rating Curve= 0 ,0
Exp/Cntr=0.3,0.1

Type RM Length L Ch R = 1 ,6246.868,354.19,1214.6,1200.65
XS GIS Cut Line= 6
      3183428.14    13774291.246     3180894.665    13774983.012
     3180715.744    13775193.917     3180575.374    13775350.684
     3180020.622    13775641.509     3178383.053    13774539.822
#Sta/Elev= 30
 1991.98   32.62 2294.45   31.45 2772.71   30.83 3127.65   31.99 3245.19   30.74
 3451.71   32.05 4137.11   32.76 4545.02   29.54 4894.79   24.24 4951.49      15
 4996.11   13.82 5001.94    12.1    5005    9.89 5018.22   10.29 5053.51   22.13
 5105.21   23.68 5240.06   24.98 5257.49   23.97 5315.85   24.46 5353.06   23.06
 5375.84   21.07 5400.53    24.3 5465.35    25.7 6572.26   26.35 6988.21    28.8
 7037.58   27.59 7062.86   28.63 7194.69   27.45 7494.23   28.95 7705.23   27.79
#Mann= 5 ,-1 , 0
 1991.98     .07       0 2294.45     .12       0 4894.79     .04       0
 5105.21     .12       0 5353.06     .07       0
#XS Ineff= 1 ,-1
    6980    7400    28.2
Permanent Ineff=
       F
#Block Obstruct= 2 ,-1
 5318.47 5419.72      24    7500 7757.72   28.31
Bank Sta=4894.79,5105.21
XS Rating Curve= 0 ,0
Exp/Cntr=0.3,0.1

Type RM Length L Ch R = 1 ,5032.265,890.28,688.4,395.74
XS GIS Cut Line= 6
      3183925.84    13773796.606     3180993.068    13774589.348
     3180578.664    13774466.239     3179897.445    13774399.054
     3179158.829    13774603.574      3178462.59    13774477.959
#Sta/Elev= 30
 1467.65   34.03 1697.92   33.75  1848.7   32.28 2033.86   32.98 2354.43   31.62
 2413.86   32.32 3006.62    31.1 3485.98   31.68  3515.6   30.95 4138.05   32.41
 4628.31   30.85 4837.49   27.88 4938.19   24.16 4994.49    8.85 5061.81   23.78
 5108.24   24.23 5156.22    26.5 5448.38   27.57 5509.29   27.15 5550.85   23.45
 5582.21   27.41 5588.33   27.43 6251.38   27.68 6354.86   26.27 6414.37   27.49
 6447.13   29.13 6518.97   27.66 6711.22   27.46 6954.25   28.99  7096.9   27.92
#Mann= 5 ,-1 , 0
 1467.65     .07       0 3006.62     .12       0 4938.19     .04       0
 5061.81     .12       0 5588.33     .07       0
#XS Ineff= 1 ,-1
    6600    6800    27.9
Permanent Ineff=
       F
#Block Obstruct= 1 ,-1
 5498.53 5596.76      25
Bank Sta=4938.19,5061.81
XS Rating Curve= 0 ,0
Exp/Cntr=0.3,0.1

Type RM Length L Ch R = 1 ,4343.861,270.64,435.52,561.82
XS GIS Cut Line= 6
      3183508.46     13773442.47     3180947.209    13773666.933
     3180392.313    13773834.782     3180320.168     13773860.91
     3178878.505    13774285.409      3178533.29    13774398.421
#Sta/Elev= 30
 1808.83   33.47 3843.16   30.98 3984.64   28.65  4019.8   30.49 4060.38   30.44
 4103.72   29.31 4448.96   28.66 4475.12   27.44 4534.58   20.05 4563.08   24.26
 4600.48   27.46 4650.08   25.99 4680.86   27.77 4818.66   26.62 4917.76   24.19
 4961.63   21.31 4995.09    8.23 5000.73    8.12 5003.31    8.16 5004.41    9.67
 5038.37   24.54 5105.47   28.91 5153.49    28.1  5208.8   29.53 5511.16   28.32
 5702.48   29.62 6112.32   27.49 6540.96   27.36 6791.96   28.85 6902.48   27.85
#Mann= 5 ,-1 , 0
 1808.83     .07       0 4060.38     .12       0 4961.63     .04       0
 5038.37     .12       0 5153.49     .07       0
#XS Ineff= 2 ,-1
 4442.81 4680.44    27.7    5350    7000      29
Permanent Ineff=
       F       F
#Block Obstruct= 1 ,-1
    3880    4050      29
Bank Sta=4917.76,5038.37
XS Rating Curve= 0 ,0
Exp/Cntr=0.3,0.1
